HEC-RAS study PETERSRN.prj: PETERSRN

--- PETERSRN.g01 (geometry) --- (continued)

Type RM Length L Ch R = 1 ,13236   ,196.5,195.2,192.3
XS GIS Cut Line= 4
2440623.90607654618972.1411131142440717.81426802618911.461974003
 2440908.5201338618804.551109855 2441005.3178081618658.632227708
#Sta/Elev= 30
       0 2130.26    35.9 2113.81    60.8 2104.74    93.9 2088.96   108.2 2080.77
   117.5 2076.16   126.6 2067.34   129.72065.697   135.8 2064.18   140.4 2063.96
     145 2064.34  150.182065.699   167.9 2068.33   183.4 2068.34   209.2 2066.96
  218.762067.239   236.3 2066.45   250.4 2068.06   262.8 2067.69   276.6 2071.15
   283.3  2071.7   291.7 2074.43   302.5 2076.16  324.492081.308   356.2 2088.35
   377.9 2095.54   448.7 2115.32  468.48 2122.02   486.4 2127.81   505.5 2133.08
#Mann= 8 ,-1 , 0
       0      .1       0    35.9      .1       0   129.7    .045       0
  150.18      .1       0  218.76      .1       0   302.5     .12       0
  324.49      .1       0  468.48      .1       0
Bank Sta=129.7,150.18
XS Rating Curve= 0 ,0
Exp/Cntr(USF)=0,0
Exp/Cntr=0.3,0.1

Type RM Length L Ch R = 1 ,13041   ,139.6,139.1,138.2
XS GIS Cut Line= 4
2440755.37754461619122.3942194842440827.61461499619076.162494447
2440976.42297995618933.1330951142441097.78125817618746.761453559
#Sta/Elev= 30
       0 2124.63    46.7 2096.32    56.2 2093.09    70.5 2090.52      80 2087.78
    95.7 2081.16  108.182074.077   117.8 2067.38   122.8 2064.58   128.9 2062.73
  138.442061.651   145.6  2060.2   151.1 2059.84   156.7 2060.02  162.412061.651
   167.8    2064   170.9 2064.19     203 2064.43   212.2 2064.93   224.7  2063.2
  228.912063.375   237.7 2064.57     253 2065.36   275.6 2068.78   319.3 2078.57
  362.452090.583   428.4 2109.07   466.7  2119.2  510.082132.202   514.6 2133.43
#Mann= 7 ,-1 , 0
       0      .1       0  108.18      .1       0  138.44    .045       0
  162.41      .1       0  228.91     .12       0  362.45      .1       0
  510.08      .1       0
#XS Ineff= 2 , 0
                          213.77         2064.94
Permanent Ineff=
       F       F
Bank Sta=138.44,162.41
XS Rating Curve= 0 ,0
Exp/Cntr(USF)=0,0
Exp/Cntr=0.3,0.1

Type RM Length L Ch R = 1 ,12902   ,189.4,195.6,199
XS GIS Cut Line= 4
2440839.17254624619242.3077562982440917.18858224619187.407582817
 2441083.3338441619008.2596482992441216.25005358618820.443265337
#Sta/Elev= 30
       0 2123.63    43.5 2099.71    87.5 2079.42     107 2072.81   145.2 2064.66
  162.23 2059.13   168.3 2057.54   174.2 2057.47     180 2057.69  185.752059.127
   193.1 2061.73   197.7 2062.24     233 2062.47   246.9 2060.38   258.2  2062.2
  281.12 2062.27   285.9  2062.7   297.8 2067.87   309.1 2071.86   348.9 2083.16
   363.2 2088.04   389.1 2094.42  415.492103.471   437.9 2111.32   449.2 2116.03
   455.1 2117.15   493.3 2128.47   527.6  2137.1  557.192146.316   569.8 2149.84
#Mann= 6 ,-1 , 0
       0      .1       0  162.23    .045       0  185.75      .1       0
  281.12     .12       0  415.49      .1       0  557.19      .1       0
#XS Ineff= 2 , 0
                          234.01         2062.58
Permanent Ineff=
       F       F
Bank Sta=162.23,185.75
XS Rating Curve= 0 ,0
Exp/Cntr(USF)=0,0
Exp/Cntr=0.3,0.1

Type RM Length L Ch R = 1 ,12706   ,175.6,171,168.3
XS GIS Cut Line= 4
2440930.19125491619353.5528446682441009.65203232619314.544826668
2441178.68677698619233.6393078542441328.93988335619066.049304595
#Sta/Elev= 30
       0 2111.97    36.3 2092.98    54.1 2084.55    71.1 2077.43    78.7 2075.12
    94.2 2068.19    98.6 2066.79   116.1 2063.17   119.1 2062.08  129.21 2055.42
   134.1    2054   142.9 2053.62   147.4 2053.71   152.6 2055.19  167.24 2057.63
   209.5  2057.2   222.8 2055.32   227.2 2055.88   231.6 2057.41     236 2058.22
  270.752060.597   292.1 2064.14   303.4 2068.71   326.1 2075.99   359.9 2088.63
   381.7 2095.14  397.19 2100.51   437.8 2112.76   455.8  2118.7     501 2135.72
#Mann= 6 ,-1 , 0
       0      .1       0  129.21    .045       0   152.6      .1       0
  167.24      .1       0  270.75     .12       0  397.19      .1       0
Bank Sta=129.21,152.6
XS Rating Curve= 0 ,0
Exp/Cntr(USF)=0,0
Exp/Cntr=0.3,0.1

Type RM Length L Ch R = 1 ,12535   ,176.1,178.6,178.4
XS GIS Cut Line= 4
2441031.32315343619544.2587104452441105.00496521619461.908450224
2441284.15289972619307.3211196312441421.40333343619172.960168743
#Sta/Elev= 30
       0  2122.6    11.1  2116.4    29.1 2108.42    82.3 2088.27   115.1 2074.23
   147.9 2062.29   164.1 2058.37   200.8 2053.21   213.1 2052.79  219.412051.415
   225.3 2050.06   231.5 2049.54   235.8 2050.07  238.622051.414   244.9 2054.16
   255.7 2051.47  270.652052.098   275.5 2052.91   289.7 2056.98   304.9 2059.55
   329.4 2066.31   352.1 2074.49   363.4 2077.39   370.6 2081.15   389.9 2088.12
   410.6  2094.6   416.4 2095.74  471.142113.058     485 2119.02   539.2 2140.31
#Mann= 5 ,-1 , 0
       0      .1       0  219.41    .045       0  238.62      .1       0
  270.65     .12       0  471.14      .1       0
Bank Sta=219.41,238.62
XS Rating Curve= 0 ,0
Exp/Cntr(USF)=0,0
Exp/Cntr=0.3,0.1

Type RM Length L Ch R = 1 ,12357   ,241.3,253,254.9
XS GIS Cut Line= 4
2441206.13686372619584.7114698532441289.93186535619531.256037779
 2441435.8507475619392.5608626682441561.54324995619259.644653187
#Sta/Elev= 30
       0 2080.73    16.2 2074.24   26.282073.273    30.7 2072.75    45.2 2068.08
    71.9  2062.8    86.1  2058.2   100.2 2055.83   117.3 2050.25     129 2049.33
   145.5 2050.39  153.032048.124     158 2046.85   172.3 2046.26   181.2  2046.7
  184.882048.121   194.3  2054.8   204.9 2060.39  247.162078.311  258.642082.749
   277.1 2088.65   291.5 2092.27   299.2  2095.2   315.3  2099.9   347.1 2111.62
   374.8 2123.22  410.162136.609   456.3 2157.34   479.4 2168.76   483.6 2171.41
#Mann= 7 ,-1 , 0
       0      .1       0   26.28      .1       0  153.03    .045       0
  184.88      .1       0  247.16     .12       0  258.64      .1       0
  410.16      .1       0
#XS Ineff= 2 , 0
          144.62 2050.34
Permanent Ineff=
       F       F
Bank Sta=153.03,184.88
XS Rating Curve= 0 ,0
Exp/Cntr(USF)=0,0
Exp/Cntr=0.3,0.1

Type RM Length L Ch R = 1 ,12104   ,121,119,113.4
XS GIS Cut Line= 4
2441297.15557239619750.8567317042441366.50315995619719.072420741
2441518.20100772619667.0617300752441684.34626957619542.813969038
#Sta/Elev= 30
       0 2082.04    25.3 2069.62    49.4 2061.33    67.8 2057.56    80.8 2053.07
    92.4 2050.54   114.4 2044.06   123.1 2043.08   135.7 2044.15     140 2043.49
   148.4 2041.77   161.6 2042.39  167.982043.423   183.7 2044.98   186.5 2046.04
   199.4  2054.6   207.6 2059.16   236.9 2067.28  267.372074.693   337.2 2092.62
   351.5 2098.23  361.052102.859   368.6 2107.12   377.2 2109.44     380  2110.9
   392.2 2119.37   410.6 2130.39   422.1 2136.42   437.1  2146.9   444.1 2150.41
#Mann= 5 ,-1 , 0
       0      .1       0     140    .045       0  167.98     .12       0
  267.37      .1       0  361.05     .12       0
Bank Sta=140,167.98
XS Rating Curve= 0 ,0
Exp/Cntr(USF)=0,0
Exp/Cntr=0.3,0.1

Type RM Length L Ch R = 1 ,11985   ,219.3,223.6,225
XS GIS Cut Line= 4
2441331.82936617619892.4413896292441440.18497172619831.762250519
2441562.98799135619746.5225074822441711.79635632619612.161556593
#Sta/Elev= 30
       0 2085.66     7.9 2083.21    17.1 2078.23    21.7 2076.32    30.8 2075.15
    41.5 2071.84    59.1 2067.42    90.4 2063.82    99.6 2061.55   113.4 2053.92
   132.7 2041.19     137  2040.4   172.6 2040.03   188.9 2038.49   195.5 2039.25
  199.722040.384   216.9 2044.69   250.2    2061  268.952068.545   284.1 2073.87
   289.5 2075.28   329.9 2083.96  357.922090.763   389.4 2096.19   406.4  2101.5
   426.2 2110.25     435 2115.19     446 2117.65   457.3 2124.99   474.2 2134.91
#Mann= 5 ,-1 , 0
       0      .1       0   172.6    .045       0  199.72      .1       0
  268.95     .12       0  357.92      .1       0
Bank Sta=172.6,199.72
XS Rating Curve= 0 ,0
Exp/Cntr(USF)=0,0
Exp/Cntr=0.3,0.1

Type RM Length L Ch R = 1 ,11761   ,150.3,149.7,147.3
XS GIS Cut Line= 4
2441453.18764439620047.0287202222441496.52988661620021.023374888
 2441708.9068735619928.5599248152441834.59937594619844.764923185
#Sta/Elev= 30
       0 2071.84    15.8 2064.22    29.8 2059.44    53.8 2059.14      66 2056.27
    85.9 2049.02    96.6 2045.87     101 2043.92  108.242037.514  110.442035.891
     114  2034.4   118.4 2034.04  131.022035.891     139 2036.69  159.192036.631
   184.5 2035.95   196.9  2036.8   223.1 2036.87   227.5 2037.47   236.2 2040.87
   240.6 2043.29     258    2055   266.6 2059.58   290.5 2065.49   299.1 2068.49
     314 2072.59   342.1 2082.21   379.9 2098.98     419 2118.82   433.2 2124.43
#Mann= 5 ,-1 , 0
       0      .1       0  108.24     .12       0  110.44    .045       0
  131.02     .12       0  159.19      .1       0
Bank Sta=110.44,131.02
XS Rating Curve= 0 ,0
Exp/Cntr(USF)=0,0
Exp/Cntr=0.3,0.1

Type RM Length L Ch R = 1 ,11611   ,174.4,170.6,165.4
XS GIS Cut Line= 4
 2441513.8667835620178.5001882952441600.55126795620139.492170295
2441778.25446106620035.4707889622441905.39170491619895.330872444
#Sta/Elev= 30
       0 2056.33   14.542052.476    31.7 2047.08      58 2041.03    84.3 2037.08
   111.5 2034.69  117.452033.111   120.8 2032.33     130 2031.42   139.3 2031.79
   148.6 2032.86   162.5 2033.24     215 2032.83   222.5 2033.25   245.9 2035.71
     255 2037.17   264.5 2037.91   278.4 2040.34   296.9 2044.74   307.2 2047.85
   334.2 2057.84   349.9 2062.71   355.5 2065.16   366.9 2068.33   379.1 2072.96
   404.4 2084.46   420.8 2092.84   454.6 2112.22   474.3 2121.78   490.2 2128.62
#Mann= 4 ,-1 , 0
       0      .1       0   14.54      .1       0  117.45    .045       0
   148.6      .1       0
Bank Sta=117.45,148.6
XS Rating Curve= 0 ,0
Exp/Cntr(USF)=0,0
Exp/Cntr=0.3,0.1

Type RM Length L Ch R = 1 ,11441   ,159.7,166.1,164.4
XS GIS Cut Line= 4
2441622.22238906 620337.42174311 2441688.6804938620285.411052443
2441838.93360017620152.4948429622441934.28653306620022.468116296
#Sta/Elev= 30
       0 2070.85    10.7 2067.25    31.1 2058.58    50.6 2051.11    71.8 2044.26
    94.2 2037.69   103.2 2034.15   113.8 2029.09   118.8 2028.28   138.6  2029.4
     150 2028.95   156.6 2029.79   167.3 2029.67   171.7  2028.8   177.9 2027.11
   183.3 2026.84  190.232028.854   203.8 2030.23   271.8 2031.06   283.2 2032.77
   297.5 2036.42   306.8 2039.49   326.7 2044.83   336.6 2046.49   351.5 2049.74
   366.4 2053.38   374.7 2055.88   397.6 2064.76     406 2067.63   446.2 2087.94
#Mann= 3 ,-1 , 0
       0      .1       0   171.7    .045       0  190.23      .1       0
Bank Sta=171.7,190.23
XS Rating Curve= 0 ,0
Exp/Cntr(USF)=0,0
Exp/Cntr=0.3,0.1

Type RM Length L Ch R = 1 ,11274   ,134.9,132.9,127.5
XS GIS Cut Line= 4
2441779.69920246620393.7666579982441834.59937594620338.866484517
2441974.73929246 620187.168636742442016.63679328620060.031392888
#Sta/Elev= 30
       0  2041.5     9.8 2038.56    32.6  2033.5      55 2027.87    63.6  2027.3
    91.9 2027.73    97.5 2027.29     106  2025.7   111.7 2025.21   131.5 2025.33
   142.7  2024.6   159.3 2024.24   164.7  2023.6   181.1 2022.92   186.5 2023.16
   189.9 2024.54   193.8 2026.65   197.4    2028   213.7 2028.42   230.6 2030.98
   254.7 2033.04   260.6 2034.48   275.9 2040.54   297.1 2049.53   326.6 2062.59
   341.1 2069.85   376.3 2086.08   398.2 2096.53   406.6  2100.9     418 2106.07
#Mann= 3 ,-1 , 0
       0      .1       0   159.3    .045       0   189.9      .1       0
Bank Sta=159.3,189.9
XS Rating Curve= 0 ,0
Exp/Cntr(USF)=0,0
Exp/Cntr=0.3,0.1

Type RM Length L Ch R = 1 ,11142   ,172.6,170.3,166.1
XS GIS Cut Line= 4
2441893.83377365620533.9065745162441951.62342994 620442.88786585
 2442020.9710175620262.2951899252442085.98438083620129.378980444
#Sta/Elev= 30
       0 2061.09    36.7 2041.72    53.9 2034.67    74.6 2030.57    98.3 2024.88
  123.612024.014   133.5 2023.73   142.1 2022.78   159.2 2023.37   167.8 2021.71
   172.3 2021.81   180.7 2020.36   184.5 2020.28   189.2 2020.31   196.9 2021.71
   203.1 2022.42   223.5 2021.44   232.1 2022.78   240.6 2022.86   261.6 2027.68
   292.1 2030.46   305.1 2034.36     314 2037.45   340.7 2049.64   358.5 2059.72
   367.4 2063.76     403 2082.86   418.8 2089.71   433.7 2097.09   449.2  2102.7
#Mann= 4 ,-1 , 0
       0      .1       0  123.61      .1       0   172.3    .045       0
   196.9      .1       0
Bank Sta=172.3,196.9
XS Rating Curve= 0 ,0
Exp/Cntr(USF)=0,0
Exp/Cntr=0.3,0.1

Type RM Length L Ch R = 1 ,10971   ,188.6,188.5,189.6
XS GIS Cut Line= 4
2442129.32662305620597.4751964422442135.10558868620496.343297924
2442150.99774417620327.3085532582442181.33731372620178.500188295
#Sta/Elev= 30
       0 2043.14    10.6 2040.07    22.6 2037.77    34.6 2033.83    50.7 2030.26
    70.7 2026.83    98.7 2022.86   110.8 2021.63   130.9  2021.2   146.9 2019.72
     163 2019.39   179.1 2016.58   191.1  2018.8  198.132016.364   212.5 2014.64
   219.3 2014.88  225.392016.365   235.3 2018.98   239.4 2021.12   247.4 2026.63
   255.4 2030.95   288.2 2043.86   311.9  2055.3   320.5 2058.52   328.9 2063.31
   345.8 2070.25   362.8 2076.47   369.6 2079.41   402.1  2095.4   422.9 2103.48
#Mann= 3 ,-1 , 0
       0      .1       0  198.13    .045       0  225.39      .1       0
#XS Ineff= 2 , 0
          153.85 2021.03
Permanent Ineff=
       F       F
Bank Sta=198.13,225.39
XS Rating Curve= 0 ,0
Exp/Cntr(USF)=0,0
Exp/Cntr=0.3,0.1

Type RM Length L Ch R = 1 ,10783   ,171,174.6,180.9
XS GIS Cut Line= 4
2442291.13766068620590.2514894052442308.47455757 620515.12493622
2442351.81679979620282.5215696282442364.81947246 620181.38967111
#Sta/Elev= 30
       0 2067.31   17.632062.095    32.2 2057.03    59.2 2048.65    72.5 2043.58
    85.5 2037.47    96.4 2029.27   101.8 2026.22   110.1 2022.73   122.1 2018.47
   134.3 2015.64   142.4 2014.51   158.7 2014.73   179.1 2013.59   187.2  2014.1
   191.3 2013.76  196.912011.438   199.4 2010.15   203.5 2009.49     213 2010.28
  218.062011.438   223.8 2014.12   227.9 2017.16   240.4 2029.63   247.3 2034.62
   276.7 2049.98  308.022068.945   321.4 2076.13   357.7 2097.14   415.7 2133.67
#Mann= 5 ,-1 , 0
       0      .1       0   17.63      .1       0  196.91    .045       0
  218.06      .1       0  308.02      .1       0
Bank Sta=196.91,218.06
XS Rating Curve= 0 ,0
Exp/Cntr(USF)=0,0
Exp/Cntr=0.3,0.1

Type RM Length L Ch R = 1 ,10608   ,203.6,207.5,212.4
XS GIS Cut Line= 4
2442367.70895528620619.1463175532442409.60645609620565.690885479
 2442529.5199929620411.1035548872442624.87292579620330.198036073
#Sta/Elev= 30
       0 2061.41    24.4 2050.16   49.35 2037.73   82.89 2022.54    90.7 2019.34
    96.8 2017.89     117 2010.37   122.1 2009.75   130.6 2010.57   137.3 2010.48
     142 2009.66  147.052007.283   152.5 2005.48   157.5 2004.95   162.6 2005.44
  168.082007.283   172.7 2008.54  185.042008.704   190.1 2009.06   196.2 2010.58
   204.7 2014.79  224.922022.879   238.5 2029.93   247.5 2033.92   275.7 2048.43
   294.8 2059.55   332.7  2079.5     344 2086.82   355.4 2091.16   388.6 2109.19
#Mann= 7 ,-1 , 0
       0      .1       0   49.35      .1       0   82.89      .1       0
  147.05    .045       0  168.08      .1       0  185.04      .1       0
  224.92      .1       0
#XS Ineff= 2 , 0
          134.06 2017.14
Permanent Ineff=
       F       F
Bank Sta=147.05,168.08
XS Rating Curve= 0 ,0
Exp/Cntr(USF)=0,0
Exp/Cntr=0.3,0.1

Type RM Length L Ch R = 1 ,10401   ,143.9,141.3,140.4
XS GIS Cut Line= 4
 2442470.2855952620707.2755434052442517.96206165620672.601749627
2442655.21249535620610.477869109 2442763.5681009 620559.91191985
#Sta/Elev= 30
       0 2040.16     6.3 2036.26    14.3 2032.43    25.3 2026.14    40.1 2020.24
    57.9 2015.25    72.9 2011.88    91.1 2009.77   108.1 2003.23   112.5 2003.19
   130.1 2005.11   134.5 2005.08   143.2 2002.79   163.6 2004.24   169.4 2003.89
   175.7 2002.55   181.7  2002.2   184.8 2002.69  187.982004.044  189.832005.654
   204.7 2020.72   208.9 2023.98   217.9  2029.3     227  2033.4   262.1 2056.04
   278.2 2067.33   284.3 2072.45   296.2 2079.09     315 2091.76   329.2 2099.25
#Mann= 4 ,-1 , 0
       0      .1       0   169.4    .045       0  187.98      .1       0
  189.83      .1       0
Bank Sta=169.4,187.98
XS Rating Curve= 0 ,0
Exp/Cntr(USF)=0,0
Exp/Cntr=0.3,0.1

Type RM Length L Ch R = 1 ,10259   ,170,170.5,170.5
XS GIS Cut Line= 4
2442512.18309602620818.520631775 2442607.5360289 620782.40209659
2442759.23387668620710.1650262192442818.46827439620692.828129331
#Sta/Elev= 30
       0 2056.17      11 2048.88    17.2 2046.22    32.7 2036.64    49.8 2027.58
    58.3 2023.64    66.9 2021.05    75.5 2017.88    88.6 2014.16    92.6 2013.15
   101.1 2011.83     110 2008.96     119 2007.47   127.7 2004.48   136.5 2000.87
  138.832000.405     146 1999.54     173 1998.96   176.4 1999.07  179.232000.406
   180.8 2001.27     191 2009.67   211.8 2025.56   260.6 2055.59   273.6  2063.9
   285.1 2069.96   291.6  2073.8   302.8 2081.36   311.2 2086.48   331.7 2101.74
#Mann= 3 ,-1 , 0
       0      .1       0  138.83    .045       0  179.23      .1       0
Bank Sta=138.83,179.23
XS Rating Curve= 0 ,0
Exp/Cntr(USF)=0,0
Exp/Cntr=0.3,0.1

Type RM Length L Ch R = 1 ,10089   ,139.1,139,138
XS GIS Cut Line= 4
2442604.64654609620949.9920998482442705.77844461620915.318306071
2442806.91034313620876.3102880712442916.71069009 620821.41011459
#Sta/Elev= 30
       0 2042.21    10.7 2035.18    23.4 2027.92    27.6 2025.74    40.3 2020.68
    58.9 2015.54      82 2010.61    99.5 2007.31   111.1 2004.69   117.3  2003.9
   123.5 2002.62   129.4 2000.56  139.011994.516   142.2 1993.26   148.2 1992.54
   150.8 1992.57   154.4 1993.13  157.381994.514   159.4 1995.75   163.7 1999.56
   176.5    2010   228.5 2047.23     233 2050.23   237.5 2052.75     242 2055.98
   250.9 2062.98   286.7 2087.88     309 2102.64   331.4    2117   338.1 2121.63
#Mann= 3 ,-1 , 0
       0      .1       0  139.01    .045       0  157.38      .1       0
Bank Sta=139.01,157.38
XS Rating Curve= 0 ,0
Exp/Cntr(USF)=0,0
Exp/Cntr=0.3,0.1

Type RM Length L Ch R = 1 ,9950    ,166.2,167.3,168.1
XS GIS Cut Line= 4
2442679.77309927621074.2398608852442769.34706653621039.566067107
2442864.69999942 620993.334342072442923.93439713620955.771065478
#Sta/Elev= 30
       0 2044.19    16.1 2034.57    38.9 2021.69    48.2 2017.27    57.5 2013.39
    63.2 2010.53    79.1 2004.87      89 2002.83    97.6 2000.44   110.9 1997.74
   119.8 1996.94   124.3 1996.07   128.7 1993.98  133.291991.026   137.6 1989.58
   145.5 1989.29   150.9 1989.64  154.881991.028   157.5 1993.28   164.3 2000.48
   170.9 2006.95   177.6 2013.06   182.1 2016.64   199.8 2028.06   213.9 2036.76
   232.9 2048.18   237.2  2050.5   243.9 2055.37     266 2068.53   272.2 2072.77
#Mann= 3 ,-1 , 0
       0      .1       0  133.29    .045       0  154.88      .1       0
Bank Sta=133.29,154.88
XS Rating Curve= 0 ,0
Exp/Cntr(USF)=0,0
Exp/Cntr=0.3,0.1

Type RM Length L Ch R = 1 ,9783    ,106.9,110,110.7
XS GIS Cut Line= 4
2442746.23120401621223.0482258472442808.35508453621198.487621922
2442955.71870809621140.697965625 2443036.6242269621111.803137477
#Sta/Elev= 30
       0 2060.21    26.4 2038.77    34.4 2032.54    39.3 2029.16    54.8 2019.31
    69.4 2011.91      78 2006.88    87.6  2002.3   103.7 1996.54   120.9 1990.82
   125.2 1989.63   133.1 1988.18  137.311986.786   142.4 1985.34   146.7    1985
   157.8 1985.65   159.6 1985.95  161.181986.784   163.9 1988.53   173.3 1998.13
   179.4 2002.77   185.6 2006.99   207.2 2020.32     232 2035.16   238.3 2038.57
   253.9 2048.95   270.8 2058.65   278.9 2063.84   296.3 2074.21     311  2083.8
#Mann= 3 ,-1 , 0
       0      .1       0  137.31    .045       0  161.18      .1       0
Bank Sta=137.31,161.18
XS Rating Curve= 0 ,0
Exp/Cntr(USF)=0,0
Exp/Cntr=0.3,0.1

Type RM Length L Ch R = 1 ,9673    ,82.1,83.5,83.6
XS GIS Cut Line= 4
2442778.01551498621316.9564173292442845.91836113621288.061589181
2443003.39517453621250.4983125882443062.62957224621230.271932884
#Sta/Elev= 30
       0 2067.11    13.8 2057.96    35.7 2045.64    39.9 2042.23    48.6 2031.91
    63.1 2020.18    78.7 2010.15    88.7 2004.48   103.4 1997.22   132.2 1985.39
   139.8 1984.13   144.6 1983.95   151.8 1982.62   156.9 1982.27   161.8 1982.46
   167.5 1984.13   169.2 1984.78   173.3 1988.04   181.7 1997.86   186.7  2002.3
   202.1 2012.73   216.8 2021.48   230.9 2030.97     235  2033.3   243.5 2039.78
   256.1 2048.24   264.6 2054.69   272.7 2059.14   285.7 2067.54   298.3 2074.02
#Mann= 3 ,-1 , 0
       0      .1       0   139.8    .045       0   167.5      .1       0
Bank Sta=139.8,167.5
XS Rating Curve= 0 ,0
Exp/Cntr(USF)=0,0
Exp/Cntr=0.3,0.1

Type RM Length L Ch R = 1 ,9589    ,86.2,83.9,82.3
XS GIS Cut Line= 4
2442818.46827438621392.0829705142442887.81586194621360.298659551
2442993.28198468621340.0722798472443043.84793394621315.511675921
#Sta/Elev= 30
       0 2061.93     4.7 2059.06    17.9  2049.9    22.3 2047.45    26.7 2044.47
    31.1 2040.46    39.9 2034.49    44.3 2031.15    53.1 2023.65    61.9 2016.62
    70.5 2010.52      80 2004.78    91.5  1996.3   103.7 1988.31   111.9 1981.13
  113.54 1980.34   115.9 1979.21     120 1978.72   126.2 1978.66   131.3 1979.06
  138.311980.343   140.4 1980.91   144.4 1983.13   156.7  1993.6   160.7 1996.66
   164.8 1999.16   189.7  2011.5     212 2024.44   216.4 2027.36   239.9 2041.39
#Mann= 3 ,-1 , 0
       0      .1       0  113.54    .045       0  138.31      .1       0
Bank Sta=113.54,138.31
XS Rating Curve= 0 ,0
Exp/Cntr(USF)=0,0
Exp/Cntr=0.3,0.1

Type RM Length L Ch R = 1 ,9505    ,98.3,97.3,96
XS GIS Cut Line= 4
2442869.03422364621472.9884893282442934.04758698621441.204178365
2443007.72939875621413.7540916252443065.51905505621383.414522069
#Sta/Elev= 30
       0 2049.98    10.8 2042.12    24.2 2033.42    37.5 2024.05    41.2 2020.83
    46.4 2016.74    59.8 2008.04    68.7 2001.03    72.4 1997.14    77.4 1991.24
    81.6 1987.22    90.2 1980.65    93.4 1979.03   96.851977.657    98.7  1976.9
   102.7 1975.92   105.8 1975.85   115.1 1976.66  117.531977.659   120.1 1978.96
   128.6 1985.82   136.9 1991.73   149.3 1999.42   163.4 2007.34   172.5  2011.7
     182 2017.42   195.1 2024.59   199.6 2027.16   208.4 2032.91   216.3 2037.66
#Mann= 3 ,-1 , 0
       0      .1       0   96.85    .045       0  117.53      .1       0
Bank Sta=96.85,117.53
XS Rating Curve= 0 ,0
Exp/Cntr(USF)=0,0
Exp/Cntr=0.3,0.1

Type RM Length L Ch R = 1 ,9408    ,115.8,116.6,117.1
XS GIS Cut Line= 4
2442908.04224164621562.5624565872442986.05827764621526.443921402
2443081.41121053621478.7674549582443117.52974572621451.317368217
#Sta/Elev= 30
       0 2045.94     4.8 2044.28    10.8 2041.13    16.2 2037.55    33.8 2026.92
    37.3 2023.93    42.6 2018.16   53.122008.664    55.9 2006.41    60.3 2003.45
    65.1 2000.77    74.1 1994.43   104.6 1977.32   110.41974.674   113.6 1973.39
     118 1972.76   124.9 1973.18  131.341974.677   135.9 1977.14   138.6 1979.17
   147.6 1987.56   154.7 1993.01   171.7 2005.01   180.7 2010.79   189.6 2017.52
   199.2 2023.11   207.7 2028.97   218.8 2035.48   229.4 2043.38   237.9 2048.74
#Mann= 4 ,-1 , 0
       0      .1       0   53.12      .1       0   110.4    .045       0
  131.34      .1       0
Bank Sta=110.4,131.34
XS Rating Curve= 0 ,0
Exp/Cntr(USF)=0,0
Exp/Cntr=0.3,0.1

Type RM Length L Ch R = 1 ,9291    ,80.6,83,84.7
XS GIS Cut Line= 4
2442961.49767372621665.1390965132443023.62155424621631.910044142
2443105.97181446621598.6809917722443159.42724653621564.007197995
#Sta/Elev= 30
       0 2016.09    11.4 2020.79    14.4 2021.22   15.662020.958    19.6  2019.4
   33.34 2010.35    37.7 2007.09    42.2 2002.83    46.9 1999.12    64.6 1988.04
    86.8 1976.08      89 1975.13    91.1 1974.31    99.7 1973.07  101.491972.487
     104 1971.53   107.4 1970.83   116.7 1970.46   122.8 1970.97   125.6 1971.54
  127.511972.484   129.9 1973.71   141.2 1982.76   147.4 1986.85   150.5 1989.22
   156.6 1994.87   160.2  1997.7   193.6  2018.9   217.4 2034.93     223 2038.96
#Mann= 5 ,-1 , 0
       0      .1       0   15.66      .1       0   33.34      .1       0
  101.49    .045       0  127.51      .1       0
Bank Sta=101.49,127.51
XS Rating Curve= 0 ,0
Exp/Cntr(USF)=0,0
Exp/Cntr=0.3,0.1

Type RM Length L Ch R = 1 ,9208    ,97.4,97.7,96.9
XS GIS Cut Line= 4
2442986.05827764621702.7023731052443045.29267535621704.147114513
 2443133.4219012621683.9207348092443230.21957549621634.799526957
#Sta/Elev= 30
       0 1999.63     4.7 2001.02     8.7 2001.58    20.7 1999.48    32.7 1994.51
    40.7 1989.79    48.7 1984.41    52.7 1982.18    56.7  1980.4    64.8 1977.75
    73.1 1975.87    85.4 1972.12   91.151970.826    97.7 1969.57   105.9 1969.13
     110 1969.18   114.1  1970.1  115.571970.825   118.2 1972.14   121.6 1974.48
   130.5 1981.73   134.6  1984.5   142.8 1989.48   151.4 1995.64   172.3 2009.07
   182.6 2016.33  198.732026.644   219.9 2040.81   245.4 2058.35   258.2 2067.72
#Mann= 4 ,-1 , 0
       0      .1       0   91.15    .045       0  115.57      .1       0
  198.73      .1       0
Bank Sta=91.15,115.57
XS Rating Curve= 0 ,0
Exp/Cntr(USF)=0,0
Exp/Cntr=0.3,0.1

Type RM Length L Ch R = 1 ,9111    ,93.6,92.6,91.4
XS GIS Cut Line= 4
2443020.73207142621805.2790130312443038.06896831621803.834271623
2443163.76147075621776.3841848832443230.21957549621746.044615327
#Sta/Elev= 30
       0 1998.01       6 1995.52      10 1993.33    18.8 1989.64    26.3 1986.03
    30.4 1982.99    34.5 1980.32    42.7 1976.22    46.7 1974.49    52.4  1972.7
   63.091968.594    67.2 1967.23    75.4  1966.8    79.9  1966.9   94.511968.592
     100 1969.32   104.1 1970.41   120.4 1970.64   124.5 1971.36   128.6 1973.91
   136.8 1981.29   140.9 1984.08   149.3 1988.82   158.1 1994.73   162.5 1997.07
   166.9 1999.85   171.3 2003.35   184.5 2012.34   215.3 2032.03   219.1 2034.75
#Mann= 3 ,-1 , 0
       0      .1       0   63.09    .045       0   94.51      .1       0
Bank Sta=63.09,94.51
XS Rating Curve= 0 ,0
Exp/Cntr(USF)=0,0
Exp/Cntr=0.3,0.1

Type RM Length L Ch R = 1 ,9018    ,149.4,142.9,135.3
XS GIS Cut Line= 4
2443009.17414016621913.6346185862443069.85327927621896.297721697
2443217.21690283621847.1765138452443269.22759349621808.168495846
#Sta/Elev= 30
       0 2015.24      10 2010.34    35.8 1996.91      64  1983.4    72.5 1979.82
    85.1 1974.03    97.8 1970.05  104.161966.429   106.2 1965.49   110.4 1964.81
   114.6 1964.59   118.9 1964.85  125.25 1966.43   131.3  1967.9   134.5 1968.08
   147.1  1967.1     161 1966.84   166.1    1967   173.7 1968.31   177.9    1970
   182.5 1972.73   188.3 1976.77   197.7 1983.88  208.471991.407   219.7 1999.12
   242.6 2012.25   251.2 2017.89   260.4 2022.68   270.4 2028.36   283.5 2036.56
#Mann= 4 ,-1 , 0
       0      .1       0  104.16    .045       0  125.25      .1       0
  208.47      .1       0
Bank Sta=104.16,125.25
XS Rating Curve= 0 ,0
Exp/Cntr(USF)=0,0
Exp/Cntr=0.3,0.1

Type RM Length L Ch R = 1 ,8875    ,128.1,127.9,126.8
XS GIS Cut Line= 4
2443156.53776372 622039.327121032443198.43526453622001.763844438
2443264.89336927621902.0766873272443293.78819742621857.289703697
#Sta/Elev= 30
       0 1996.29     4.7 1993.43    12.6 1987.99    24.5 1980.35    30.2 1977.85
    35.2 1974.79    41.5 1971.59    45.9 1969.75      50  1968.5    56.3 1967.26
    67.2 1965.62      79 1964.16   87.741962.367    98.2 1960.74   104.7 1960.69
   107.8 1960.76   112.6 1961.54  115.031962.366   124.9 1965.22     127 1965.95
   128.9 1966.93   131.8 1968.92   142.2 1978.23   151.1 1985.31   156.6  1988.8
   162.4 1991.86   180.6 2002.31   194.2 2010.72     218 2024.06   229.4 2031.29
#Mann= 3 ,-1 , 0
       0      .1       0   87.74    .045       0  115.03      .1       0
Bank Sta=87.74,115.03
XS Rating Curve= 0 ,0
Exp/Cntr(USF)=0,0
Exp/Cntr=0.3,0.1

Type RM Length L Ch R = 1 ,8747    ,161.5,161.4,159.1
XS GIS Cut Line= 4
2443237.44328253622154.9064336222443285.11974898622114.453674215
 2443348.6883709621987.3164303632443379.02794046621926.637291253
#Sta/Elev= 30
       0 2016.31     9.4 2011.71    15.1 2007.95    22.7 2002.31    43.3 1987.01
    54.9  1979.4    59.4 1976.74    72.4 1970.01    84.7 1964.07    90.2 1962.22
    96.2 1961.35   120.1 1961.71   124.6 1960.63  128.541958.515   133.6 1956.74
   137.7 1956.49   143.9    1957   146.7 1957.64   148.61958.517   151.5  1960.2
   155.8  1964.6   158.8 1967.17   164.5 1971.31   173.8 1976.89   187.3 1984.25
   191.6 1987.01   197.6    1990   236.3 2013.14   263.2 2028.61   272.5 2034.47
#Mann= 4 ,-1 , 0
       0      .1       0    22.7      .1       0  128.54    .045       0
   148.6      .1       0
#XS Ineff= 2 , 0
          119.22 1962.01
Permanent Ineff=
       F       F
Bank Sta=128.54,148.6
XS Rating Curve= 0 ,0
Exp/Cntr(USF)=0,0
Exp/Cntr=0.3,0.1

Type RM Length L Ch R = 1 ,8586    ,138.5,138.2,137.5
XS GIS Cut Line= 4
2443409.36751001622257.4830735482443425.25966549622202.582900066
2443474.38087335622071.1114319932443480.15983898621990.205913178
#Sta/Elev= 30
       0 2015.06    12.9  2004.9    40.2 1985.18    45.2 1981.26    57.2 1971.17
    69.6 1959.75    74.5 1957.38    78.2 1956.87   89.371956.895   112.3  1958.4
  118.45 1955.29   120.9 1954.03   125.1 1953.44   133.7 1953.76     138 1954.46
  140.421955.291   146.5 1957.03   150.8 1959.11   164.3 1967.45   166.9  1969.3
   176.4 1977.21   189.2 1984.59  200.841992.349   209.8 1997.09   229.8 2009.34
   241.8 2015.45   249.9 2020.61   257.9 2023.98   266.4 2029.88   278.6 2037.07
#Mann= 5 ,-1 , 0
       0      .1       0   89.37      .1       0  118.45    .045       0
  140.42      .1       0  200.84      .1       0
Bank Sta=118.45,140.42
XS Rating Curve= 0 ,0
Exp/Cntr(USF)=0,0
Exp/Cntr=0.3,0.1

Type RM Length L Ch R = 1 ,8448    ,104.5,102.1,100.3
XS GIS Cut Line= 4
2443536.50475386622308.0490228072443556.73113357622247.369883696
2443591.40492735622146.2379851782443597.18389298622029.213931178
#Sta/Elev= 30
       0 2029.26    13.9 2018.31    26.5 2005.61    47.6 1986.73    51.8 1983.67
    59.6 1978.79    78.5 1964.79    84.8 1960.89    89.8 1957.92    94.1 1955.97
  100.051955.442   106.8 1954.64  111.761952.327   115.2 1951.08   125.8 1950.68
   132.1 1950.82   136.4 1951.63  137.641952.328   140.6    1954     149 1961.37
   157.5 1966.54   163.5 1971.45   169.8 1976.07   182.2 1984.31   206.3 1999.29
   234.3 2015.59   254.3 2026.33   263.6 2030.79   274.3 2036.62     288  2043.5
#Mann= 4 ,-1 , 0
       0      .1       0  100.05      .1       0  111.76    .045       0
  137.64      .1       0
Bank Sta=111.76,137.64
XS Rating Curve= 0 ,0
Exp/Cntr(USF)=0,0
Exp/Cntr=0.3,0.1

Type RM Length L Ch R = 1 ,8345    ,175.4,173.8,171.6
XS GIS Cut Line= 4
2443650.63932505622336.9438509552443662.19725631622280.598936066
 2443680.9788946622162.130140659 2443679.5341532622050.885052289
#Sta/Elev= 30
       0 2017.34    10.3 2010.15    38.8 1987.67    51.1 1977.07    71.4 1962.49
    75.4 1958.75    79.5 1955.52    83.5 1954.17      91 1952.91   98.021949.657
    99.7 1948.91   103.8 1948.18   107.8 1948.13   115.9 1948.15     120 1948.52
  123.861949.658   132.1 1951.08   132.9 1951.49   137.7 1954.59   172.6 1980.31
   176.7 1982.63   184.7 1986.51   196.7 1994.14   204.7 1997.98   212.7 2003.27
   248.7 2024.21   264.7 2034.33   272.7 2037.66   276.7 2039.76   288.7 2047.85
#Mann= 3 ,-1 , 0
       0      .1       0   98.02    .045       0  123.86      .1       0
Bank Sta=98.02,123.86
XS Rating Curve= 0 ,0
Exp/Cntr(USF)=0,0
Exp/Cntr=0.3,0.1

Type RM Length L Ch R = 1 ,8172    ,137.5,145.1,147.6
XS GIS Cut Line= 4
2443832.67674238622368.7281619182443841.34519083622284.933160288
2443838.45570801  622150.57220942443809.56087986622037.882379623
#Sta/Elev= 30
       0 2043.41      30 2029.09   61.772015.391    70.2 2011.11    78.3 2006.14
    82.3 1999.69    90.3 1976.35    94.3 1966.96    98.3 1962.58   106.3 1958.39
   118.3  1950.3   122.3 1948.78   130.3 1947.83  143.951943.708   150.3 1942.12
   154.3 1941.89   162.3 1942.13  167.391943.707   170.3  1945.4   178.3 1952.37
   186.3 1958.24   194.3 1965.57   214.3 1981.31   218.6 1984.24   230.7 1990.88
   267.9 2014.83   280.2 2025.19   317.4 2051.08   329.7 2058.55     335 2062.46
#Mann= 4 ,-1 , 0
       0      .1       0   61.77      .1       0  143.95    .045       0
  167.39      .1       0
Bank Sta=143.95,167.39
XS Rating Curve= 0 ,0
Exp/Cntr(USF)=0,0
Exp/Cntr=0.3,0.1

Type RM Length L Ch R = 1 ,8027    ,101.8,107.9,114.7
XS GIS Cut Line= 4
2443919.36122683622387.509800214 2443952.5902792622309.493764214
2443988.70881438 622222.809279772443968.48243468622094.227294511
#Sta/Elev= 30
       0 2032.48    18.1 2024.57    35.5 2015.11    39.8 2010.68    44.1 2004.06
    48.5 1996.41    52.8 1990.54    57.9 1985.59    65.9 1978.33    80.1 1967.12
    96.3 1955.63  107.791945.333   109.8 1943.94     118 1941.53  124.851938.377
     131 1936.73   139.6 1936.69   146.6 1937.41  149.731938.377   161.3  1945.8
     170 1952.67   190.8 1959.73   198.9 1963.94   215.1 1970.52   227.2 1976.76
   243.3 1987.97   259.6 1997.35     288 2014.81   304.1 2025.22   308.9 2029.09
#Mann= 4 ,-1 , 0
       0      .1       0  107.79      .1       0  124.85    .045       0
  149.73      .1       0
Bank Sta=124.85,149.73
XS Rating Curve= 0 ,0
Exp/Cntr(USF)=0,0
Exp/Cntr=0.3,0.1

Type RM Length L Ch R = 1 ,7919    ,97.9,103.9,108.6
XS GIS Cut Line= 4
2443978.59562453622391.8440244362444021.93786675622355.725489251
2444094.17493712 622300.825315772444175.08045594622238.701435252
#Sta/Elev= 30
       0  2002.8     1.5 2000.84     5.4 1994.63     7.7 1991.66    15.8 1983.53
      21 1979.47    47.1 1962.73    51.5 1959.21    57.4 1952.58    60.4 1948.21
    62.5 1945.66    67.5 1940.93    72.5 1937.92    82.6 1936.46   85.311935.533
    92.6 1933.67   103.3 1934.17   107.7 1934.76  110.171935.532   117.3 1938.64
   132.8 1947.95   152.9 1956.74     168 1965.43   183.2 1973.56   194.6 1980.58
   203.3 1984.12     216 1990.97   223.5 1994.01   235.7 2000.03   249.2 2007.92
#Mann= 3 ,-1 , 0
       0      .1       0   85.31    .045       0  110.17      .1       0
Bank Sta=85.31,110.17
XS Rating Curve= 0 ,0
Exp/Cntr(USF)=0,0
Exp/Cntr=0.3,0.1

Type RM Length L Ch R = 1 ,7815    ,104.9,115.2,120.6
XS GIS Cut Line= 4
2444014.71415971622446.7441979182444063.83536757622429.407301029
2444164.96726608622403.4019556952444260.32019897 622367.28342051
#Sta/Elev= 30
       0 1987.67     4.3 1984.97     8.5  1981.7      17 1973.82    21.2 1970.64
    46.7 1953.94    50.9 1950.38    59.2 1942.46    63.4 1939.27    67.5 1936.59
    71.6 1934.81      73 1934.52    75.7 1934.02    82.8 1933.63   85.941932.982
    92.3 1931.77   100.5 1931.12   104.7 1931.24   108.8 1931.83     113 1932.98
     117 1935.41   129.4 1945.73   148.5 1959.39   158.3 1965.42   169.2 1972.62
   176.9 1976.55  194.781987.663   226.9 2007.85   238.9 2015.87   258.5 2027.75
#Mann= 4 ,-1 , 0
       0      .1       0   85.94    .045       0     113      .1       0
  194.78      .1       0
Bank Sta=85.94,113
XS Rating Curve= 0 ,0
Exp/Cntr(USF)=0,0
Exp/Cntr=0.3,0.1

Type RM Length L Ch R = 1 ,7700    ,96.1,103.4,109.8
XS GIS Cut Line= 4
2444024.82734957622511.7575612512444065.28010897622511.757561251
2444169.30149031622543.5418722132444258.87545756622563.768251917
#Sta/Elev= 30
       0 1969.97     9.9 1963.32      42 1946.15    50.3 1942.12    62.9    1935
    67.1  1932.1    71.3 1930.28    83.8 1930.05   85.731929.587    92.2 1928.19
   104.7 1927.91   111.4  1928.4   113.1 1928.71  114.671929.589   117.3 1931.06
     121 1934.61   125.6 1938.25   130.6 1943.96     134  1946.8   142.4 1951.86
   146.5 1954.87   167.1 1967.35   187.6 1981.63   195.8 1986.77   200.1 1990.41
  209.212001.824   212.2 2004.87   220.4 2011.18   236.7 2020.24   241.1 2021.41
#Mann= 4 ,-1 , 0
       0      .1       0   85.73    .045       0  114.67      .1       0
  209.21      .1       0
Bank Sta=85.73,114.67
XS Rating Curve= 0 ,0
Exp/Cntr(USF)=0,0
Exp/Cntr=0.3,0.1

Type RM Length L Ch R = 1 ,7596    ,82.7,81.6,79.9
XS GIS Cut Line= 4
2443982.92984875622569.5472175472444042.16424645622585.439373028
2444098.50916134622644.6737707322444140.40666216622679.347564509
#Sta/Elev= 30
       0 1961.44     8.1 1959.22    23.8 1951.85    32.9 1949.11    37.1 1947.44
    74.4 1931.29    79.7 1929.47    91.1 1927.99   96.141925.951    99.5 1924.66
   102.4 1924.04   107.5 1923.89   114.4 1924.59  121.421925.951   133.5 1928.48
   136.3 1929.52   139.2 1931.03   143.4 1934.44   150.5    1942   153.3 1944.32
   161.9 1949.91   164.2 1952.07  165.681954.268   167.6 1957.68   173.2 1968.99
   176.1 1973.47   177.9 1975.47   179.7 1976.63   184.2 1978.28   197.5 1982.14
#Mann= 4 ,-1 , 0
       0      .1       0   96.14    .045       0  121.42      .1       0
  165.68      .1       0
Bank Sta=96.14,121.42
XS Rating Curve= 0 ,0
Exp/Cntr(USF)=0,0
Exp/Cntr=0.3,0.1

Type RM Length L Ch R = 1 ,7515    ,140.7,132.6,118
XS GIS Cut Line= 4
2443936.69812371622604.221011324 2443972.8166589622638.894805102
2444042.16424645622698.1292028062444092.73019571622727.024030954
#Sta/Elev= 30
       0  1972.6    14.7  1962.8    32.7  1950.5    45.8 1942.28    51.4 1939.05
    63.1 1933.12    74.7 1928.11    80.9 1926.11    91.2 1924.16   96.271922.514
    99.9 1921.29   102.5 1920.82   105.3 1920.51   108.2 1920.48   115.7    1921
  123.321922.513   126.3 1923.32   130.1 1925.42   139.6 1935.42   141.9 1937.47
   145.2 1939.19  150.591941.579   156.9 1945.85   158.9 1946.89     165 1948.99
   168.6 1950.85   171.6 1951.91   174.5  1952.7   177.4 1953.21   199.5 1955.41
#Mann= 4 ,-1 , 0
       0      .1       0   96.27    .045       0  123.32      .1       0
  150.59      .1       0
Bank Sta=96.27,123.32
XS Rating Curve= 0 ,0
Exp/Cntr(USF)=0,0
Exp/Cntr=0.3,0.1

Type RM Length L Ch R = 1 ,7382    ,120.4,109.3,93.5
XS GIS Cut Line= 4
2443831.23200097622783.3689458422443897.69010571 622779.03472162
2444003.15622845622770.3662731762444081.17226445 622740.02670362
#Sta/Elev= 30
       0 1983.97   30.611959.775    43.6 1949.06    63.6 1934.25    71.7 1928.57
    75.7 1926.39    83.7 1922.69    87.7 1921.16    91.7 1920.28   95.48 1918.27
    99.8  1916.6   103.8 1916.41   115.8    1917   123.8 1918.63   131.9 1918.83
   135.9 1918.13   139.9 1918.17   145.6  1921.5     156 1929.22   160.4 1932.09
     164 1934.09     168 1934.87   179.6 1940.13   189.1 1943.43   197.7 1947.13
   210.6 1951.22   221.1 1953.39   227.3 1954.41  231.031954.625   256.1 1953.46
#Mann= 5 ,-1 , 0
       0      .1       0   30.61      .1       0   95.48    .045       0
   123.8      .1       0  231.03      .1       0
Bank Sta=95.48,123.8
XS Rating Curve= 0 ,0
Exp/Cntr(USF)=0,0
Exp/Cntr=0.3,0.1

Type RM Length L Ch R = 1 ,7273    ,100.1,97.8,94.2
XS GIS Cut Line= 4
2443965.59295186622958.1826561382443988.70881438622903.282482657
2444037.83002223622805.0400669532444063.83536757622764.587307546
#Sta/Elev= 30
       0  1979.2    15.6 1968.78    20.9 1965.01      34 1956.84    51.3 1943.05
    64.5 1934.38    77.9 1926.36    86.8 1920.25    91.3 1917.69    95.8 1915.72
   100.1 1914.76   104.7 1914.26  107.041913.817   113.7 1912.13     118 1911.69
   122.6 1912.15  130.741913.818   131.6 1914.06   135.9 1916.31   138.9 1917.35
   140.5 1917.75     145 1918.12   149.4 1918.94   153.6 1920.76   171.6 1929.72
   176.7 1932.42     191 1940.45   205.2 1947.25   215.81951.574   217.5 1952.28
#Mann= 4 ,-1 , 0
       0      .1       0  107.04    .045       0  130.74      .1       0
   215.8      .1       0
Bank Sta=107.04,130.74
XS Rating Curve= 0 ,0
Exp/Cntr(USF)=0,0
Exp/Cntr=0.3,0.1

Type RM Length L Ch R = 1 ,7175    ,97.7,96.3,93.8
XS GIS Cut Line= 4
2444085.50648868622992.8564499162444094.17493712622933.622052212
2444117.29079964622822.3769638422444118.73554105622783.368945842
#Sta/Elev= 30
       0 1978.65       6 1974.01    10.1 1971.21    18.2 1965.75    30.3 1958.03
   34.071955.438    46.5 1946.47    54.5  1940.9    62.7 1935.66    74.9 1927.01
    91.3 1914.36    95.3 1911.68   97.961910.501    99.4 1909.86   103.5 1908.76
   107.6 1908.43   111.7 1908.61   115.8 1909.26  120.391910.502   123.9 1911.61
     128  1912.6   140.5 1913.46   144.4 1914.22   148.4 1915.46     154  1918.1
   165.8 1925.39   173.5  1929.6     197 1939.31   208.9 1943.51   212.5 1945.05
#Mann= 4 ,-1 , 0
       0      .1       0   34.07      .1       0   97.96    .045       0
  120.39      .1       0
Bank Sta=97.96,120.39
XS Rating Curve= 0 ,0
Exp/Cntr(USF)=0,0
Exp/Cntr=0.3,0.1

Type RM Length L Ch R = 1 ,7079    ,121.1,123.3,124.6
XS GIS Cut Line= 4
2444195.30683564622988.5222256932444198.19631845622939.401017842
2444201.08580127622838.2691193242444198.19631845622789.147911472
#Sta/Elev= 30
       0 1975.34     5.6 1971.79    13.7 1967.14    29.7 1956.04    31.3  1954.7
    37.7 1949.03    41.7 1944.16    45.7 1938.11    53.7 1930.82    57.7 1926.29
    61.7 1922.55    65.7 1919.85    77.7 1913.23    81.7 1911.35   90.961908.171
    93.7    1907    97.7 1906.22   105.7 1905.93   109.7  1906.6  114.42 1908.17
   121.7 1910.27   125.7 1912.27   133.8  1916.7   141.8 1922.34  145.371924.469
   165.8 1936.41   173.8 1942.24   186.1 1948.53   193.6 1954.24   199.6 1957.58
#Mann= 4 ,-1 , 0
       0      .1       0   90.96    .045       0  114.42      .1       0
  145.37      .1       0
Bank Sta=90.96,114.42
XS Rating Curve= 0 ,0
Exp/Cntr(USF)=0,0
Exp/Cntr=0.3,0.1

Type RM Length L Ch R = 1 ,6955    ,130.4,138.7,148.2
XS GIS Cut Line= 4
2444306.55192401 623001.524898362444312.33088964622949.514207694
2444326.77830371622864.2744646572444329.66778653622792.037394287
#Sta/Elev= 30
       0 1992.89    14.7 1986.58    18.7 1984.13    22.8 1979.54    26.8 1971.17
    30.8  1960.1    34.8 1950.72    38.9 1944.16    42.9 1939.52    50.9  1934.1
      55 1931.58      59 1928.28    63.6 1924.01    78.21913.301    87.4 1906.96
   90.341905.526    91.5 1904.96    95.6 1904.13   103.7 1903.89   111.8 1904.07
   115.8 1904.94  117.031905.529     124 1908.76   132.1 1911.31   143.9 1917.92
   160.2 1926.14     167 1930.15   176.2 1934.84   196.2 1946.05   211.1 1953.46
#Mann= 4 ,-1 , 0
       0      .1       0    78.2      .1       0   90.34    .045       0
  117.03      .1       0
Bank Sta=90.34,117.03
XS Rating Curve= 0 ,0
Exp/Cntr(USF)=0,0
Exp/Cntr=0.3,0.1

Type RM Length L Ch R = 1 ,6817    ,112.7,114.9,114.5
XS GIS Cut Line= 4
 2444362.8968389623039.088174953 2444401.9048569622989.966967101
2444484.25511712622922.0641209532444530.48684216622852.716533398
#Sta/Elev= 30
       0 1992.97     8.6 1987.44    10.5 1985.81    14.3 1980.34    17.1 1975.19
    20.7  1969.3    28.5 1959.48    30.9 1956.98    41.1 1948.93      57 1937.89
    63.8 1931.43      69 1925.07    79.7 1913.86    84.6 1909.63    91.1 1905.07
    98.81900.635   105.3 1898.75   110.5 1898.56  122.881900.637     126 1901.05
     128 1901.89   130.9 1903.44   136.7 1908.07   141.6  1910.1   149.3 1912.13
   168.2  1921.8   202.1  1941.2   215.2 1947.92   226.2 1954.95   252.8  1970.9
#Mann= 3 ,-1 , 0
       0      .1       0    98.8    .045       0  122.88      .1       0
Bank Sta=98.8,122.88
XS Rating Curve= 0 ,0
Exp/Cntr(USF)=0,0
Exp/Cntr=0.3,0.1

Type RM Length L Ch R = 1 ,6702    ,151.6,147.6,141.8
XS GIS Cut Line= 4
2444442.35761631 623118.54895236 2444481.3656343623066.538261693
2444565.16063593623002.9696397682444609.94761956622919.174638138
#Sta/Elev= 30
       0 1994.15     9.6 1987.98    14.6 1984.26    17.2 1980.62    20.6  1974.8
    27.3 1959.23    29.6 1954.41    31.5 1951.21      34 1948.05    49.6 1936.53
    71.5 1918.34    74.3 1915.26    81.8 1905.46    85.7 1902.62    91.4 1899.59
   98.211897.172   105.7 1895.85     117 1895.34     122 1895.99  126.271897.174
     132  1899.7   142.1 1902.01   148.5 1905.17     160 1911.56   189.2 1929.59
   203.9  1939.1   224.6 1951.47   236.4 1957.46   245.3 1961.42   265.2 1971.94
#Mann= 3 ,-1 , 0
       0      .1       0   98.21    .045       0  126.27      .1       0
Bank Sta=98.21,126.27
XS Rating Curve= 0 ,0
Exp/Cntr(USF)=0,0
Exp/Cntr=0.3,0.1

Type RM Length L Ch R = 1 ,6554    ,130.7,125.8,118.3
XS GIS Cut Line= 4
2444583.94227423623205.2334368042444609.94761956623164.780677397
2444663.40305164623080.9856757672444685.07417275622976.964294434
#Sta/Elev= 30
       0 1972.32     3.7 1962.22     7.5 1952.55     9.5 1949.12    12.3 1945.35
    17.1  1942.4    21.1 1939.56    27.4  1933.3    31.3 1929.98    36.1 1926.84
    49.6 1917.03    58.7 1909.11    69.3 1900.81   78.091893.414    79.3 1892.67
    83.5 1891.69    88.3 1891.64    97.8 1892.06  103.721893.412     112 1896.39
   122.5 1898.65   131.4 1902.41   147.5 1911.19     166 1920.32   185.9 1931.32
     196 1938.53   210.9 1947.07   229.9 1956.62   247.7 1966.03   253.7 1968.88
#Mann= 3 ,-1 , 0
       0      .1       0   78.09    .045       0  103.72      .1       0
Bank Sta=78.09,103.72
XS Rating Curve= 0 ,0
Exp/Cntr(USF)=0,0
Exp/Cntr=0.3,0.1

Type RM Length L Ch R = 1 ,6428    ,172.5,171.8,170.8
XS GIS Cut Line= 4
2444739.97434623623260.1336102852444747.19805327623206.678178211
2444755.86650171623095.4330898412444747.19805327622988.522225694
#Sta/Elev= 30
       0 1963.76     1.3  1961.8     3.6 1959.92    37.6 1936.21    49.6 1926.15
    53.7    1922    57.7  1915.9    65.8  1900.3    73.8 1892.81   79.011889.897
    81.8 1889.08    93.8 1887.88   101.9  1888.6  103.941889.894   105.9 1891.09
   109.9 1892.21   125.9 1892.34     130 1892.63     134  1893.7     138  1895.8
   145.6 1901.09     158 1911.92   174.1 1923.69   182.1 1927.44   194.2 1935.37
   210.2 1944.55   222.3 1949.79   230.4 1953.96   258.4 1964.65   272.8 1971.16
#Mann= 3 ,-1 , 0
       0      .1       0   79.01    .045       0  103.94      .1       0
Bank Sta=79.01,103.94
XS Rating Curve= 0 ,0
Exp/Cntr(USF)=0,0
Exp/Cntr=0.3,0.1

Type RM Length L Ch R = 1 ,6257    ,144.4,151.2,157.6
XS GIS Cut Line= 4
2444904.67486667623290.4731798412444920.56702216623231.238782137
2444922.01176356623091.098865619 2444909.0090909623011.638088212
#Sta/Elev= 30
       0 1958.89    20.3 1944.98    24.4 1941.06    38.9 1929.23    45.1 1923.64
    61.3 1912.07    77.7  1900.8    93.7 1890.76    97.7 1888.51  103.671886.092
   105.7 1885.29   109.7 1884.46   117.7 1884.29   121.7 1884.58  129.31 1886.09
   133.7 1886.52   137.7 1887.38   141.7  1888.6   145.7 1890.64   153.7 1896.81
   173.7  1913.9   177.7 1916.73   189.7  1924.2   205.7 1935.83   218.4 1943.93
     226 1947.91   238.2 1955.17   266.5 1969.48   274.6  1972.7     282 1976.21
#Mann= 3 ,-1 , 0
       0      .1       0  103.67    .045       0  129.31      .1       0
Bank Sta=103.67,129.31
XS Rating Curve= 0 ,0
Exp/Cntr(USF)=0,0
Exp/Cntr=0.3,0.1

Type RM Length L Ch R = 1 ,6105    ,144.1,139.5,133
XS GIS Cut Line= 4
2445011.58573082623323.7022322112445030.36736912623281.804731396
2445092.49124964623174.8938672482445117.05185356623076.651451545
#Sta/Elev= 30
       0 1954.33     9.7 1947.35    18.1 1940.68    24.2 1936.24    27.2 1933.64
      36 1927.06    44.7 1919.27    53.9 1909.86    67.8 1897.66    74.7 1892.76
    80.5 1887.97      86    1884    89.3  1882.7   92.541881.838   100.2 1880.37
   104.8 1879.92   109.8 1879.85   112.7 1880.33  118.191881.839   121.5 1882.57
   123.3 1883.26   130.3 1889.39   134.2 1892.31   147.8 1900.26   160.3 1908.06
   186.1 1923.42     219 1941.98     252 1957.23   260.3 1960.22   270.8 1964.52
#Mann= 3 ,-1 , 0
       0      .1       0   92.54    .045       0  118.19      .1       0
Bank Sta=92.54,118.19
XS Rating Curve= 0 ,0
Exp/Cntr(USF)=0,0
Exp/Cntr=0.3,0.1

Type RM Length L Ch R = 1 ,5966    ,131.9,132.1,132.3
XS GIS Cut Line= 4
2445180.62047549 623374.268181472445186.39944112623309.254818137
 2445183.5099583623198.0097297672445199.40211378 623079.54093436
#Sta/Elev= 30
       0 1955.39    15.4 1943.48    19.5 1939.43    23.5 1934.88    30.9 1928.09
    39.5 1920.96    43.5 1916.91    55.6 1906.26    67.6 1893.61    75.6 1885.91
    79.6 1880.89   83.02  1877.9    87.6 1875.95    91.6 1875.63    95.6 1876.18
  102.161877.903   107.6 1879.01   111.6  1879.2   127.7 1879.05   135.7 1882.49
   143.7 1886.84   156.9 1895.77   179.7 1910.37   187.8 1914.57     212 1930.16
   240.2 1947.24   248.3 1950.91   264.5 1959.46   276.6 1965.02   296.1 1972.58
#Mann= 3 ,-1 , 0
       0      .1       0   83.02    .045       0  102.16      .1       0
Bank Sta=83.02,102.16
XS Rating Curve= 0 ,0
Exp/Cntr(USF)=0,0
Exp/Cntr=0.3,0.1

Type RM Length L Ch R = 1 ,5834    ,139.5,139.7,138.8
XS GIS Cut Line= 4
2445309.20246075623403.1630096182445316.42616778623338.149646285
2445317.87090919623219.6808508782445303.42349512623127.217400804
#Sta/Elev= 30
       0 1959.52     4.3 1954.26    12.3 1947.24    23.4 1938.49    32.5 1929.98
    44.5 1919.42    48.6 1915.47    56.6 1905.88    60.6  1902.2    72.7  1892.9
    80.7 1887.37    92.7 1877.51      981874.533   100.7  1873.5   104.7 1872.68
   108.7  1872.5   112.7  1872.8  120.31 1874.53   128.7  1875.2   132.7 1876.29
   148.7 1882.62   160.7 1888.47   168.7 1892.96   192.8 1907.43   205.1 1916.01
   225.2  1931.1   229.3 1933.89   248.3 1943.71   261.6 1951.09   277.5    1958
#Mann= 3 ,-1 , 0
       0      .1       0      98    .045       0  120.31      .1       0
Bank Sta=98,120.31
XS Rating Curve= 0 ,0
Exp/Cntr(USF)=0,0
Exp/Cntr=0.3,0.1

Type RM Length L Ch R = 1 ,5694    ,150.2,151.4,151.4
XS GIS Cut Line= 4
2445452.23186008623406.0524924332445455.12134289623330.925939248
2445453.67660149623231.2387821372445406.00013504623121.438435175
#Sta/Elev= 30
       0 1954.91     7.2 1948.18    15.2 1937.82    19.2 1933.23    23.2  1925.7
    27.2 1918.99    51.2 1902.54    79.5    1881    91.2 1873.35    95.2  1871.9
  106.791870.222   111.2 1868.77   115.2 1868.57   131.2 1869.25  135.231870.226
   143.2 1877.45   155.2 1884.95   159.2 1888.37   163.2 1890.97   175.3 1893.66
   179.6  1895.8   185.3  1900.1   197.1 1907.01   218.9 1921.71   227.6  1926.1
   236.3  1931.2   244.3  1934.4   258.1 1941.59   282.7 1951.74   294.6 1957.23
#Mann= 3 ,-1 , 0
       0      .1       0  106.79    .045       0  135.23      .1       0
Bank Sta=106.79,135.23
XS Rating Curve= 0 ,0
Exp/Cntr(USF)=0,0
Exp/Cntr=0.3,0.1
